HEC-RAS study WFGRNBRRRV.prj: WFGRNBRRRV

--- WFGRNBRRRV.g01 (geometry) --- (continued)

Type RM Length L Ch R = 1 ,83560   ,331.2,360.9,395.6
XS GIS Cut Line= 3
2313288.94032186618125.422875694 2313134.5137365617994.071527226
2312529.23252261617878.695342761
#Sta/Elev= 30
       0 3059.15    31.9 3053.46   121.8 3040.82     148 3031.34   158.5 3029.07
   173.2 3027.48     188 3028.49   208.9 3027.57   229.7 3025.01   245.8 3019.45
     254 3019.87   271.6 3018.39   343.6 3020.66   359.9 3019.43   408.7 3020.98
   463.8  3018.1   473.9 3017.07   498.3 3018.18   502.4 3019.42   514.6 3026.98
   522.7 3028.57   533.8 3027.99   544.1 3024.42   555.3 3023.39   632.7 3026.92
     653 3028.34   681.5 3032.23     758 3038.34   780.1 3042.47   818.9 3046.45
#Mann= 10 ,-1,0
       0      .1       0      70     .06       0  302.73      .1       0
   463.8    .045       0   498.3      .1       0  502.73     .07       0
  572.73     .06       0  602.73      .1       0  702.73     .12       0
  802.73      .1       0
#XS Ineff= 2 , 0
          254.57 3024.09
Permanent Ineff=
       F       F
Bank Sta=463.8,498.3
XS Rating Curve= 0 ,0
Exp/Cntr(USF)=0,0
Exp/Cntr=0.3,0.1

Type RM Length L Ch R = 1 ,83199   ,674.4,641.6,612.9
XS GIS Cut Line= 4
2313312.01555875618123.6478574722313224.22149988617991.003409245
2313093.71237778617662.965220498 2312707.7349788617432.045843453
#Sta/Elev= 30
       0 3060.28    65.3 3047.86    74.9 3048.36    86.7 3045.56   151.7 3037.08
     161 3035.34   173.9 3028.69   199.8 3029.09   234.2 3026.24   245.8 3024.25
   259.1 3018.66   268.7  3016.9   305.3 3016.62   320.3 3015.89   339.1 3016.63
   386.4 3019.14   458.1 3017.82   549.5 3023.73   575.8  3023.9   593.1 3025.58
   619.5  3025.1   718.7 3030.12   733.3 3027.44   741.5 3027.36   793.6 3031.59
   849.5 3031.44     874 3035.85   891.5 3036.27   920.7 3034.47   961.9 3037.67
#Mann= 8 ,-1,0
       0      .1       0     120     .06       0  229.07      .1       0
   305.3    .045       0   339.1     .12       0  582.11      .1       0
  692.11     .06       0  812.11      .1       0
Bank Sta=305.3,339.1
XS Rating Curve= 0 ,0
Exp/Cntr(USF)=0,0
Exp/Cntr=0.3,0.1

Type RM Length L Ch R = 1 ,82557   ,447.8,449.3,439.6
XS GIS Cut Line= 3
2313779.20871753617665.9139216622313133.32285012617586.790889128
2312681.88408975617355.064967111
#Sta/Elev= 30
       0 3057.27    71.6  3039.4    95.7 3028.22   115.9 3026.89     128 3019.02
     132 3018.28   180.4 3018.77   204.6 3015.31   337.5  3017.1   351.43013.234
   377.8 3012.12   384.8  3013.2   389.9 3015.18   418.1 3016.53   458.4 3014.54
   499.5 3017.08   526.9 3014.62   563.2 3018.06   635.2 3020.97   701.5 3021.69
   855.7 3027.24   873.2 3030.81   894.8 3027.21   960.8 3031.42   993.7 3030.81
  1065.9 3038.84  1097.1  3039.5  1125.2 3052.51  1144.8 3059.88  1158.2 3062.71
#Mann= 11 ,-1,0
       0      .1       0      60     .06       0     150      .1       0
     350     .12       0   351.4    .045       0   384.8     .12       0
     650      .1       0  870.71     .06       0  980.71      .1       0
  990.71     .12       0 1090.71      .1       0
#XS Ineff= 2 , 0
          203.32 3026.54
Permanent Ineff=
       F       F
Bank Sta=351.4,384.8
XS Rating Curve= 0 ,0
Exp/Cntr(USF)=0,0
Exp/Cntr=0.3,0.1

Type RM Length L Ch R = 1 ,82108   ,441.5,456.2,476.1
XS GIS Cut Line= 5
2313883.73863919617483.2122867852313663.19259137617291.626831101
2313448.11518364617326.8616997482313099.78244155617383.177730039
2312935.57689943617265.125980187
#Sta/Elev= 30
       0 3065.79    47.1 3054.68   121.3 3039.91   126.6 3038.42   145.7 3028.24
   151.4 3026.69   179.8 3026.31   222.3 3018.38   267.7 3017.02   292.1 3017.83
   314.13013.095   323.6 3011.22   338.93012.802     356 3015.14   408.7 3015.51
   425.5 3014.07   465.4 3013.92   492.7 3014.94   501.9 3016.64   514.1 3015.23
   530.3  3015.4   542.4 3013.68   611.3 3014.64   676.2 3016.89   692.4 3016.37
   858.5 3023.47   911.7 3022.49   931.4 3024.72  1005.3 3028.39  1065.2 3048.75
#Mann= 7 ,-1,0
       0      .1       0      80     .06       0     210      .1       0
   314.1    .045       0   338.9      .1       0  942.94     .06       0
 1062.94     .12       0
#XS Ineff= 2 , 0
          277.08 3024.49
Permanent Ineff=
       F       F
Bank Sta=314.1,338.9
XS Rating Curve= 0 ,0
Exp/Cntr(USF)=0,0
Exp/Cntr=0.3,0.1

Type RM Length L Ch R = 1 ,81652   ,617.3,637.5,640.8
XS GIS Cut Line= 2
2313993.62255621617310.6895115472313051.08788004616833.209609683
#Sta/Elev= 30
       0 3047.88    77.9 3034.09   145.1 3024.24   158.6 3025.27   180.4 3022.34
   338.5 3018.73   390.6 3018.98   433.8 3016.86     450 3019.92   463.6  3015.4
   481.4 3012.78   573.6 3013.22   594.5 3012.75   602.5 3010.74   612.3 3009.75
     6293010.708   638.3  3013.1   656.3 3013.79     737 3012.29   853.1 3013.89
   868.3 3025.01     885 3026.13   889.5 3027.99   897.3 3034.32   951.6 3069.12
   979.1 3085.26  1010.5 3109.29    1024 3114.37  1032.9 3114.28  1056.6 3119.14
#Mann= 10 ,-1,0
       0      .1       0      80     .06       0     300     .12       0
     410      .1       0   602.5    .045       0     629      .1       0
     630     .08       0     820     .06       0     960     .12       0
    1040      .1       0
#XS Ineff= 2 , 0
          450.45 3023.27
Permanent Ineff=
       F       F
Bank Sta=602.5,629
XS Rating Curve= 0 ,0
Exp/Cntr(USF)=0,0
Exp/Cntr=0.3,0.1

Type RM Length L Ch R = 1 ,81014   ,327.1,345.9,363.9
XS GIS Cut Line= 3
2314164.02430557617092.3622701742313324.44068631616604.232258975
 2313095.4633356616636.182586981
#Sta/Elev= 30
       0 3090.17    98.8 3068.17   161.8 3048.83   175.6 3039.17   197.3 3037.66
     208 3031.18   221.9 3026.36   268.2 3019.19   428.1 3016.83   587.7 3018.15
   629.1  3015.6   672.2 3014.95   735.5 3017.07   744.8 3016.47   758.6 3012.59
   795.7 3012.99   803.93010.663   809.8 3008.95   832.7 3008.49   851.2 3010.77
   882.9 3023.13   892.8 3025.16   906.7 3025.34   920.6 3035.47   938.5 3042.24
   983.6 3052.06  1060.3 3058.63  1076.4 3063.01  1124.9 3082.12  1202.4 3097.56
#Mann= 10 ,-1,0
       0      .1       0     110     .06       0     280     .12       0
     500      .1       0     510     .12       0     620      .1       0
     740     .06       0   803.9    .045       0   851.2     .06       0
     960      .1       0
#XS Ineff= 2 , 0
          578.14 3023.87
Permanent Ineff=
       F       F
Bank Sta=803.9,851.2
XS Rating Curve= 0 ,0
Exp/Cntr(USF)=0,0
Exp/Cntr=0.3,0.1

Type RM Length L Ch R = 1 ,80668   ,173,170.8,171.3
XS GIS Cut Line= 4
2314175.48407235 616859.596137882313766.48250507 616565.42060322
2313647.49400281616380.579962935 2313189.5393014616126.752357111
#Sta/Elev= 30
       0 3056.18    52.8 3042.19      78 3040.74   101.5 3028.42   168.5 3025.21
   206.1 3017.89   408.3 3015.71   437.7 3012.77     482 3016.24   540.4 3016.09
   560.6 3010.93   565.9 3007.85   589.7 3007.09   606.9 3010.92     623 3010.58
   641.7 3019.03   680.1 3030.68   740.3 3037.81   759.4 3036.41   771.9 3024.69
   777.7 3023.44   791.5 3023.65   814.3 3033.67   937.8 3029.54   993.4  3024.1
  1060.7 3026.33  1077.2 3028.71  1102.4 3038.94  1175.6 3055.38  1247.2 3080.38
#Mann= 8 ,-1,0
       0     .06       0      70     .12       0   560.6    .045       0
   606.9      .1       0  643.81     .12       0  743.63     .06       0
  863.63     .12       0  993.63      .1       0
#XS Ineff= 2 , 0
          351.16 3028.76
Permanent Ineff=
       F       F
Bank Sta=560.6,606.9
XS Rating Curve= 0 ,0
Exp/Cntr(USF)=0,0
Exp/Cntr=0.3,0.1

Type RM Length L Ch R = 1 ,80498   ,185.1,183.5,183.6
XS GIS Cut Line= 4
 2314315.0330748616590.8766874982313957.55220902616545.740214545
2313771.58994045  616262.28316442313320.22521092615996.880703436
#Sta/Elev= 30
       0 3064.73      19 3060.28    39.2 3051.27    75.5 3050.51   160.1 3034.08
   236.8 3024.59   286.9 3012.99   466.2 3015.19   504.5 3011.84   518.9 3009.07
  534.25 3009.98   566.8 3008.33   574.3  3009.9   581.6 3013.81   600.2 3016.14
   693.9 3015.82   740.4 3013.59     759 3019.34   786.8 3022.44   872.1 3020.89
   893.5 3018.89     926 3019.45   939.3 3023.22   961.9 3026.42  1046.7 3034.41
  1069.9 3038.38  1102.4 3041.24  1162.7 3051.02  1185.9  3051.3  1222.9 3058.72
#Mann= 8 ,-1,0
       0     .06       0     100     .12       0  480.32      .1       0
  534.25    .045       0   574.3      .1       0  719.33     .06       0
  869.33     .12       0  919.33      .1       0
#XS Ineff= 2 , 0
          320.93 3022.37  744.19         3025.78
Permanent Ineff=
       F       F
Bank Sta=534.25,574.3
XS Rating Curve= 0 ,0
Exp/Cntr(USF)=0,0
Exp/Cntr=0.3,0.1

Type RM Length L Ch R = 1 ,80314   ,353.7,308.3,265.8
XS GIS Cut Line= 5
2314286.00281829616434.1692098742314057.45171374  616362.7469897
2313984.24393806616253.828103935 2313919.5373119616154.346602395
2313438.95345403615774.811736203
#Sta/Elev= 30
       0  3040.2    73.2  3034.2    94.1 3031.42   131.8 3022.98   152.8 3023.83
   169.5 3020.38   260.6 3014.46  292.79 3009.85   299.1 3009.28   337.7 3009.87
   347.4 3013.13   361.8 3014.95   390.5 3015.87   422.2 3010.41   451.5 3011.28
   475.3 3014.16   605.8  3014.3   613.9 3015.19   620.7 3018.77   632.1 3021.13
   640.7 3020.35   652.1 3015.53   657.8 3014.64   820.4 3017.89   884.9 3021.71
   917.2  3021.3     988 3030.96  1028.8 3043.25  1074.7 3052.49  1101.7 3056.36
#Mann= 8 ,-1,0
       0     .06       0      70      .1       0  292.79    .045       0
   337.7     .12       0  480.69      .1       0  489.36     .06       0
  739.36     .12       0  859.36      .1       0
#XS Ineff= 2 , 0
                          799.34          3026.2
Permanent Ineff=
       F       F
Bank Sta=292.79,337.7
XS Rating Curve= 0 ,0
Exp/Cntr(USF)=0,0
Exp/Cntr=0.3,0.1

Type RM Length L Ch R = 1 ,80006   ,119.4,123.4,127.8
XS GIS Cut Line= 3
2314296.71615132616018.1347773622314011.02727063616066.344775979
2313512.85728491615707.448119607
#Sta/Elev= 30
       0  3059.8    12.7 3055.25    37.1 3054.56    49.2 3050.13    89.8 3042.12
   130.4 3031.54   146.6 3022.49  161.46 3009.53   166.9 3007.06   199.3 3007.57
   211.7  3009.5   231.8 3013.88     280 3013.99     308 3012.95   352.4 3014.97
   430.2 3012.76   446.1 3019.47   455.9 3020.47   464.5 3019.05   475.7 3014.74
   510.4  3012.6   549.6 3013.23   572.3 3015.66     586  3014.7   687.6 3017.84
   746.8 3021.28   763.9 3019.55   825.5 3025.03   835.5 3028.48   903.7 3044.17
#Mann= 8 ,-1,0
       0     .06       0      80     .12       0  161.46    .045       0
   211.7     .12       0     280      .1       0  309.73     .06       0
  519.73     .12       0  649.73      .1       0
#XS Ineff= 2 , 0
                          453.52         3022.76
Permanent Ineff=
       F       F
Bank Sta=161.46,211.7
XS Rating Curve= 0 ,0
Exp/Cntr(USF)=0,0
Exp/Cntr=0.3,0.1

Type RM Length L Ch R = 1 ,79883   ,174.1,197.5,224.4
XS GIS Cut Line= 4
2314326.02845411615973.6129194682314175.93521729615922.151492583
2313903.57411714615937.552022945 2313559.5423689615677.527423678
#Sta/Elev= 30
       0 3062.51    23.1 3057.59    33.3 3054.16    52.7 3053.23    61.2 3049.79
    74.2 3046.55   124.5 3036.23   158.7 3028.36   214.7 3009.11   222.5 3006.51
   234.6 3005.92   258.6 3008.83   297.8  3013.7   306.7 3014.04   318.7 3012.73
   326.7  3013.8   338.7 3012.01   370.8 3014.54   406.8 3013.88   422.7 3019.05
   435.7  3020.2   442.7 3018.85     452  3014.4   467.5 3012.26     536 3012.83
   652.3 3013.62     734 3015.71   750.5 3019.12   801.7 3024.71   862.7 3034.37
#Mann= 7 ,-1,0
       0     .06       0   124.5     .12       0   214.7    .045       0
   258.6     .12       0   318.7     .06       0     536     .12       0
   652.3      .1       0
#XS Ineff= 2 , 0
                          432.11         3023.57
Permanent Ineff=
       F       F
Bank Sta=214.7,258.6
XS Rating Curve= 0 ,0
Exp/Cntr(USF)=0,0
Exp/Cntr=0.3,0.1

Type RM Length L Ch R = 1 ,79685   ,168.4,168.1,167.9
XS GIS Cut Line= 4
2314379.60146047615869.4410098662314173.34456057615787.903777764
2314082.00730845615698.7942634922313674.33128065615371.316798543
#Sta/Elev= 30
       0 3062.65      51 3050.76    63.9 3048.94    70.7 3049.99    85.4 3049.22
      94 3043.86    98.3 3042.61     180 3028.02   201.5 3022.77   235.9 3011.76
   247.2 3011.95   255.7 3010.01   264.1  3011.1   271.5 3011.81   290.5 3008.03
   311.6  3006.1  319.45 3008.01   334.5 3017.05     346 3018.84   354.7 3017.49
   366.1 3010.21   371.1 3008.81   409.5 3009.98   431.5 3009.55   676.2 3011.38
   684.7 3012.95   731.4  3028.5   772.9  3037.7   807.1 3043.57   872.3 3059.43
#Mann= 9 ,-1,0
       0      .1       0    70.7     .06       0     180     .12       0
   264.1     .06       0   290.5    .045       0  319.45     .06       0
   409.5      .1       0   431.5     .12       0   731.4      .1       0
#XS Ineff= 2 , 0
                          345.92         3021.28
Permanent Ineff=
       F       F
Bank Sta=290.5,319.45
XS Rating Curve= 0 ,0
Exp/Cntr(USF)=0,0
Exp/Cntr=0.3,0.1

Type RM Length L Ch R = 1 ,79517   ,359,359.4,359.7
XS GIS Cut Line= 2
 2314447.3659773615822.017945332 2313797.5969773615184.908945332
#Sta/Elev= 30
       0 3075.85    90.5 3059.53   116.5 3053.93   133.3 3046.52   161.2 3045.76
     232 3029.03   275.4 3017.05   284.6 3016.51   295.8 3007.72   305.5 3005.26
   316.8  3005.5  321.82 3007.65   336.6  3016.6   345.1 3018.51   356.4 3018.12
   370.6 3011.31     419 3006.26     464 3006.57   486.2 3008.34     512 3008.03
   581.5    3007   601.1 3009.08     624 3010.71   650.6 3009.33   712.8 3008.99
   732.6  3013.1   789.6 3044.08   823.9 3059.19   835.3 3061.37     910 3087.21
#Mann= 10 ,-1,0
       0      .1       0    90.5     .06       0     232     .12       0
   295.8    .045       0  321.82     .06       0   370.6      .1       0
     464     .12       0     512      .1       0   601.1     .12       0
   650.6      .1       0
#XS Ineff= 2 , 0
                          347.61         3022.61
Permanent Ineff=
       F       F
Bank Sta=295.8,321.82
XS Rating Curve= 0 ,0
Exp/Cntr=0.3,0.1

Type RM Length L Ch R = 1 ,79158   ,517.8,488.7,454
XS GIS Cut Line= 2
2314808.35592035615682.9978014762314286.50056293615155.817389381
#Sta/Elev= 30
       0 3124.28   120.8 3081.14   170.8  3059.6   176.8 3058.17   196.6 3049.36
   236.2  3034.9   250.3 3027.22   267.3 3026.21   272.7 3024.74   284.5 3016.18
   295.2 3010.88   312.1 3008.88   385.3 3007.67     420 3008.43   430.3 3008.97
   445.5 3006.61   468.1 3004.42   475.3  3006.8   496.4 3016.16   509.1 3018.31
   516.2 3017.77   524.7 3015.33   542.9 3005.08   564.3 3004.53   587.9 3006.13
   610.4 3014.66   638.6 3029.11   654.8 3032.26   700.5 3047.83   741.8 3062.91
#Mann= 7 ,-1,0
       0      .1       0   170.8     .06       0   312.1      .1       0
     420     .06       0   445.5    .045       0   475.3     .06       0
   700.5      .1       0
#XS Ineff= 2 , 0
                          506.14         3025.33
Permanent Ineff=
       F       F
Bank Sta=445.5,475.3
XS Rating Curve= 0 ,0
Exp/Cntr(USF)=0,0
Exp/Cntr=0.3,0.1

Type RM Length L Ch R = 1 ,78669   ,384.5,366.8,349.2
XS GIS Cut Line= 3
2315165.13458309615090.1417151472314600.67878832615154.042371158
2314439.15213007615077.716587589
#Sta/Elev= 30
       0 3163.27     158 3082.62   230.4 3054.13   250.5 3041.17   260.4 3040.98
   274.7 3037.83   294.8 3025.16   310.9 3010.64     323 3004.87   339.1 3003.27
   360.8 3004.74   371.3 3006.83   419.8 3005.96   447.8 3010.69   504.2 3011.76
   581.9  3041.9     604 3052.94   608.4  3051.3   612.9 3046.13   617.2 3039.73
   626.1 3021.71   629.2 3018.98   643.8  3018.3   648.3 3023.42   653.2 3033.25
   661.5 3041.86   668.2 3056.36   670.4 3060.71   679.2 3069.13   746.7  3086.5
#Mann= 5 ,-1,0
       0      .1       0   260.4     .06       0     323    .045       0
   360.8      .1       0   668.2     .06       0
Bank Sta=323,360.8
XS Rating Curve= 0 ,0
Exp/Cntr(USF)=0,0
Exp/Cntr=0.3,0.1

Type RM Length L Ch R = 1 ,78302   ,475.6,475.7,476.5
XS GIS Cut Line= 2
2314891.78177681614637.5120683982314405.42678384614997.840767574
#Sta/Elev= 30
       0 3130.22    62.4 3102.12    89.1 3087.67   139.6 3063.86   153.8 3054.91
   178.7 3052.52   196.8  3039.8   205.4 3036.57   213.9 3031.63   245.4 3019.09
   258.4 3009.66   271.1 3003.45   281.7 3001.76   299.7 3001.95   307.1 3003.36
   318.1 3006.08     343 3006.32   357.9 3009.23   379.8 3008.51   402.7 3010.03
   442.7 3017.12   468.5 3017.13   472.4 3018.81   482.4 3026.98   496.7 3033.16
   523.5 3047.61   537.2 3052.32     572 3071.06     582 3074.84   605.3 3087.04
#Mann= 9 ,-1,0
       0      .1       0      70     .06       0     230      .1       0
   271.1    .045       0   307.1      .1       0     350     .06       0
     470      .1       0     570     .06       0     590      .1       0
Bank Sta=271.1,307.1
XS Rating Curve= 0 ,0
Exp/Cntr(USF)=0,0
Exp/Cntr=0.3,0.1

Type RM Length L Ch R = 1 ,77826   ,418.4,444.3,468.3
XS GIS Cut Line= 2
2314620.20398877614264.7582416642314089.47354023614637.512068398
#Sta/Elev= 30
       0 3075.58    34.3 3068.91    80.5 3057.46    92.9 3053.07   112.5 3053.06
   166.2 3035.47   175.5 3034.36   185.8 3028.65   215.1 3016.76   224.9 3016.32
     264 3005.95     293 3007.36     308  3006.5   327.8  3002.7   347.8 3003.54
   355.7 3001.81   379.3 3003.58   393.7 3011.47   400.9 3013.43   428.2 3012.96
   479.1 3034.78     520 3054.47   532.8  3064.2   540.3 3067.64   548.7 3074.29
   586.6 3098.46   597.6 3101.01     611 3111.32   620.8 3114.16   648.6  3130.3
#Mann= 6 ,-1,0
       0      .1       0      10     .06       0     130      .1       0
   347.8    .045       0   379.3     .06       0     490      .1       0
#XS Ineff= 2 , 0
                          406.98         3028.29
Permanent Ineff=
       F       F
Bank Sta=347.8,379.3
XS Rating Curve= 0 ,0
Exp/Cntr(USF)=0,0
Exp/Cntr=0.3,0.1

Type RM Length L Ch R = 1 ,77382   ,471.7,478.6,474.6
XS GIS Cut Line= 3
     2314783.829      614182.3222314151.59917801614042.880963846
2313996.77707737614176.547204928
#Sta/Elev= 30
       0 3130.09    65.2 3111.18    73.4 3107.62   106.1 3099.78   141.6 3088.19
   155.3 3086.26   178.5 3078.19   257.7 3056.25   278.2 3045.34   306.9  3044.1
   323.2 3035.94   380.6 3019.09   474.8 3008.06     528 3005.55   544.4 3006.24
   564.5 3003.12   577.2 3001.09   589.5 3001.51   593.6 3003.28   605.9 3010.39
   638.6 3012.87   642.7 3015.66   654.3 3027.66     677 3044.23   715.4  3063.2
   747.1 3074.49   762.9    3076   787.6 3082.66   834.6 3085.44     852 3085.09
#Mann= 6 ,-1,0
       0      .1       0     180     .06       0     280      .1       0
   564.5    .045       0   593.6     .06       0  687.42      .1       0
Bank Sta=564.5,593.6
XS Rating Curve= 0 ,0
Exp/Cntr=0.3,0.1

Type RM Length L Ch R = 1 ,76904   ,372.1,373,371.5
XS GIS Cut Line= 2
2314735.58017323613826.3287406962314135.62401401613616.876590436
#Sta/Elev= 30
       0  3100.9    16.1 3096.43    72.7 3073.98   147.7 3040.48   160.6 3030.75
   164.6 3029.47   181.6 3028.41   194.3 3018.99   198.3 3017.18   228.2 3011.38
   245.1  3001.8   258.3 3000.39     262 2999.36   287.5 2999.05   295.9  3000.4
   329.8 3006.06   363.7 3004.76   418.8 3006.15   433.8  3010.6   456.9 3012.55
   495.1 3027.62   516.3 3040.47   524.7 3046.84   533.2 3049.36     550 3060.03
   558.6 3065.49   584.6 3077.44   597.1 3084.47   613.7 3089.48   635.5 3099.04
#Mann= 7 ,-1,0
       0      .1       0     110     .06       0     240      .1       0
   258.3    .045       0   295.9      .1       0     410     .06       0
     550      .1       0
Bank Sta=258.3,295.9
XS Rating Curve= 0 ,0
Exp/Cntr(USF)=0,0
Exp/Cntr=0.3,0.1

Type RM Length L Ch R = 1 ,76531   ,397.4,400.1,403.5
XS GIS Cut Line= 3
2314879.35664926613487.3002601912314364.60136472613309.798437936
2314224.37492514613164.246943688
#Sta/Elev= 30
       0 3102.95    83.8 3072.78   126.9  3054.9   159.9 3038.34   176.8 3026.36
     198 3023.87   210.7 3014.68   227.6 3005.47   265.7 3002.73   299.5 3002.85
   309.4 2999.95   328.2 2997.84     344 2999.85     344 2999.86     363 3004.63
   392.6 3002.15   419.5 3003.01   439.2 3011.12   456.1 3011.82   469.8 3024.91
   476.1 3028.97   548.1 3057.57   573.9 3070.77   593.3 3077.14     616 3088.59
   628.7 3091.78   650.9 3103.54   700.8 3123.06   723.5 3130.07   746.6 3140.34
#Mann= 8 ,-1,0
       0      .1       0      80     .06       0     180      .1       0
   309.4    .045       0     344      .1       0     390     .07       0
     490     .06       0   564.5      .1       0
Bank Sta=309.4,344
XS Rating Curve= 0 ,0
Exp/Cntr(USF)=0,0
Exp/Cntr=0.3,0.1

Type RM Length L Ch R = 1 ,76130   ,239.8,251.7,261.8
XS GIS Cut Line= 2
2315039.10828929613146.4967614632314419.62692962612885.569082749
#Sta/Elev= 30
       0 3087.84    55.2 3075.33      90 3064.72   107.4 3061.32   137.7 3050.65
   150.8 3048.06   165.1 3041.36   181.1 3031.13   185.5 3029.68   207.2 3029.08
   250.6 3009.28   281.6 3002.49   351.4 3002.83   359.1 2999.85   366.7 2997.73
   409.4 2999.92   433.9  3009.7   454.6 3010.68   467.6 3014.69   488.8 3029.17
     498 3031.21   506.7 3038.36   516.3 3042.68   545.7 3063.45   554.4 3066.34
   571.8 3082.05   590.8 3091.13     614 3107.98   658.6 3133.46   672.2 3139.63
#Mann= 6 ,-1,0
       0      .1       0     120     .06       0     250      .1       0
   359.1    .045       0   409.4     .06       0     470      .1       0
Bank Sta=359.1,409.4
XS Rating Curve= 0 ,0
Exp/Cntr(USF)=0,0
Exp/Cntr=0.3,0.1

Type RM Length L Ch R = 1 ,75879   ,210.6,212.9,209.7
XS GIS Cut Line= 2
2315087.71723974612996.9748640152314652.04169668612664.861540207
#Sta/Elev= 30
       0 3065.45    56.6  3049.9    69.8 3047.61      95 3040.78   110.8 3033.04
   135.2 3031.42   145.3  3025.3   170.4 3014.45   190.7  3007.7   225.8 3001.11
     266 2999.08   293.5 3000.55   301.2 2998.92   304.9 2998.07   326.4 2997.53
   336.4 2998.96   349.4 3003.04   364.8 3004.17     382 3009.75   401.8 3009.68
   424.8 3015.56   428.5 3018.28     442  3031.6   472.2 3048.63   482.3 3056.35
   497.4 3065.79   507.5 3073.21   517.5 3078.99   532.6 3091.45   547.8  3099.5
#Mann= 6 ,-1,0
       0     .06       0     150      .1       0   301.2    .045       0
   336.4      .1       0     350     .06       0     480      .1       0
Bank Sta=301.2,336.4
XS Rating Curve= 0 ,0
Exp/Cntr(USF)=0,0
Exp/Cntr=0.3,0.1

Type RM Length L Ch R = 1 ,75666   ,205.5,204.8,200.5
XS GIS Cut Line= 3
2315197.08491109612913.9693743092315083.48374485612734.692533833
2314794.15577457612528.790420018
#Sta/Elev= 30
       0 3073.41      36 3062.92    67.2 3052.43   109.9 3044.07   119.3 3036.36
   124.1 3034.02   160.7 3034.61   175.2 3031.15   190.4 3024.61   204.1 3015.89
   218.6 3008.75     231 3004.02   250.7 3001.56   298.9 3004.78   330.4 2999.13
   352.8 2997.71   359.1 2999.16   368.5 3000.31     393 3000.12   412.7 3001.39
   428.7 3008.87     448 3010.69   456.3 3012.98   468.1 3022.61   488.2 3033.01
     506 3044.57   515.8 3046.07   519.7 3047.83   559.8 3074.05   567.4 3078.04
#Mann= 7 ,-1,0
       0      .1       0      10     .06       0     170      .1       0
   330.4    .045       0   359.1      .1       0  432.24     .06       0
  552.24      .1       0
Bank Sta=330.4,359.1
XS Rating Curve= 0 ,0
Exp/Cntr(USF)=0,0
Exp/Cntr=0.3,0.1

Type RM Length L Ch R = 1 ,75461   ,263.8,257.7,232.3
XS GIS Cut Line= 3
2315230.56168009612841.6315351372315105.57279479612502.375989312
2314882.37835674612384.529326025
#Sta/Elev= 30
       0 3057.82    42.7 3049.55    55.9 3041.18    81.5 3042.27   102.8 3031.72
   136.2 3030.03     158    3025   179.8 3022.41   210.9 3017.02   226.4 3015.77
   257.7 3010.19   273.3 3006.26   279.5 3006.01   291.9 3009.56   326.2 3008.17
   398.4 3001.94   419.5 2998.28   426.5 2997.31   457.9 2998.43   467.2 3001.24
   480.7 3009.41   498.8 3011.26   512.4 3022.05   530.5  3033.5   558.8 3056.97
   573.6 3066.77   584.8 3071.32   593.8  3077.1   602.9 3084.59   613.9 3089.76
#Mann= 7 ,-1,0
       0      .1       0      40     .06       0     150      .1       0
   419.5    .045       0   457.9      .1       0  471.55     .06       0
  591.55      .1       0
Bank Sta=419.5,457.9
XS Rating Curve= 0 ,0
Exp/Cntr(USF)=0,0
Exp/Cntr=0.3,0.1

Type RM Length L Ch R = 1 ,75203   ,301.3,271.2,242.4
XS GIS Cut Line= 3
2315397.66197024612289.1629599742315028.45817995 612223.48728574
2314884.68170392612246.562522633
#Sta/Elev= 30
       0 3047.52    13.7 3047.37    25.9 3045.98    42.1 3038.85    97.8 3022.06
   147.8 3008.91     160 3006.87   180.3 3000.31     191    3000   204.8 3001.03
   220.9 3000.14   235.8 3000.55     244 2997.35   253.4 2996.54     290 2996.38
   308.2 2997.28   314.3 2998.07   338.7 3004.16   350.9 3009.16   371.2 3010.13
     375 3012.45   391.5 3029.04   407.7 3040.29   415.8 3044.56     428 3053.54
   440.1 3058.96   453.5 3069.04   488.7 3089.48     513 3100.45   520.6 3102.86
#Mann= 4 ,-1,0
       0      .1       0     244    .045       0   308.2     .06       0
     395      .1       0
Bank Sta=244,308.2
XS Rating Curve= 0 ,0
Exp/Cntr(USF)=0,0
Exp/Cntr=0.3,0.1

Type RM Length L Ch R = 1 ,74932   ,125.9,126.3,128.8
XS GIS Cut Line= 3
2315382.46564871611803.878875394 2315070.9102726612032.046663917
2314921.58069286612096.597821655
#Sta/Elev= 30
       0 3061.27     7.8 3062.91    22.7 3061.58    36.9 3054.35    49.6  3053.4
    76.7  3046.9    91.3 3045.14   126.8 3035.37   177.2 3025.72   222.9 3014.79
   248.7 3011.85   260.7    3012   274.5 3008.45   290.4 2996.12   295.4 2994.84
   306.8 2994.61   323.1 2994.75   328.8 2996.06     340 2998.06   349.9 2997.52
   379.6 3001.87   415.3 3001.08   419.7 3002.11   432.7 3008.76     453 3009.98
   477.3 3027.91   515.5  3050.4   524.2 3051.52     533 3055.59   548.9 3059.84
#Mann= 5 ,-1,0
       0     .06       0     100      .1       0   290.4    .045       0
   328.8      .1       0  456.17     .06       0
#XS Ineff= 2 , 0
                           382.3         3005.79
Permanent Ineff=
       F       F
Bank Sta=290.4,328.8
XS Rating Curve= 0 ,0
Exp/Cntr(USF)=0,0
Exp/Cntr=0.3,0.1

Type RM Length L Ch R = 1 ,74806   ,164.3,157.4,151.7
XS GIS Cut Line= 2
2315282.39796313611737.9836614792314874.54479353 612006.09431082
#Sta/Elev= 30
       0 3054.32    12.2 3051.04    34.9 3041.49    42.2 3039.25    45.7 3038.82
    55.3 3040.55    60.1 3040.52    74.5 3037.79    90.6 3033.32     115 3030.11
   133.9 3025.92   154.1 3020.32   218.1 3012.23   263.9 2995.69   270.7 2994.36
   285.1 2994.27   299.4 2995.66   328.2  2999.2   352.1 3003.64   366.5 3008.88
   385.2 3007.68   393.8 3008.69   404.8 3012.79   419.1 3019.53   428.5 3024.82
   434.3 3025.97   442.9 3030.56   457.4 3034.13   474.7  3040.1   488.1 3042.02
#Mann= 6 ,-1,0
       0     .06       0     100      .1       0   263.9    .045       0
   299.4      .1       0     330     .06       0     450      .1       0
Bank Sta=263.9,299.4
XS Rating Curve= 0 ,0
Exp/Cntr(USF)=0,0
Exp/Cntr=0.3,0.1

Type RM Length L Ch R = 1 ,74648   ,193.6,185.2,179.2
XS GIS Cut Line= 2
2315163.35956486611570.2805798452314776.40559235611937.709351911
#Sta/Elev= 30
       0 3081.55    15.8 3073.25    26.9 3073.48    38.3 3071.81    46.7 3065.48
    59.6 3058.92    91.3 3046.41   108.8 3039.07   120.4 3035.88   213.7 2996.34
   230.7 2998.18   250.5 2994.15   259.8 2993.33   290.1  2994.3   307.8 2996.71
   321.2 2996.73   335.3 3000.03   351.9 2999.65     358 3000.83   370.2 3007.71
   380.6  3007.8   397.6 3004.99   440.2 3018.03   462.7 3020.22     474 3016.15
   478.8  3015.8   484.3 3017.27     491 3021.13   510.8 3030.26   533.6 3034.56
#Mann= 6 ,-1,0
       0     .06       0    91.3      .1       0   250.5    .045       0
   290.1      .1       0   351.9     .06       0     491      .1       0
Bank Sta=250.5,290.1
XS Rating Curve= 0 ,0
Exp/Cntr(USF)=0,0
Exp/Cntr=0.3,0.1

Type RM Length L Ch R = 1 ,74463   ,333.1,280.8,225.8
BEGIN DESCRIPTION:
xs 4
END DESCRIPTION:
XS GIS Cut Line= 3
2314931.41674945 611473.122838192314770.55035985611741.233487531
2314760.80088169611911.849355294
#Sta/Elev= 30
       0 3074.75     9.4 3073.03    22.8 3062.35    37.4  3053.6    57.8 3043.14
      70 3038.67    79.4 3032.56    95.7 3024.86   121.3 3006.66   135.3 2998.33
     140 2996.49   156.9 2993.71   172.7 2992.45   183.2  2993.7   200.7 2994.91
     238 3000.62   276.5 3000.26   289.3 3005.54   296.9 3007.24   307.9  3006.6
   320.6 3002.37   352.8 3004.33   392.7  3011.6   412.1 3011.47   420.8 3008.17
   428.6 3008.25   436.8 3011.15   452.8 3019.48   476.9 3028.05   483.6 3028.93
#Mann= 5 ,-1,0
       0     .06       0      70      .1       0   156.9    .045       0
   183.2     .06       0     300      .1       0
#XS Ineff= 2 , 0
                          252.11         3007.39
Permanent Ineff=
       F       F
Bank Sta=156.9,183.2
XS Rating Curve= 0 ,0
Exp/Cntr(USF)=0,0
Exp/Cntr=0.5,0.3

Type RM Length L Ch R = 1 ,74182   ,91.2,103,118.2
BEGIN DESCRIPTION:
xs 3
END DESCRIPTION:
XS GIS Cut Line= 6
2314459.01078347611340.6711471192314452.28362415611403.880220531
2314481.63127844611447.9017019612314510.57071404611479.563518505
2314753.74821052 611685.465632322314744.87311941611914.442983027
#Sta/Elev= 30
       0 3034.63    28.5 3033.24    52.8 3022.69    63.6 3015.55      76 3016.16
    98.8 3014.21   118.2  3014.2   126.2 3017.53   136.2 3018.54   156.1  3010.9
   170.2 3007.81   193.3 2997.46   212.8 2993.01     227 2992.45   249.8 2991.62
   265.2 2992.54     286 2994.97   343.3 2996.45   359.2 2994.02   375.2  2999.1
   388.8 3000.85     478 3000.59   493.8 3006.06   501.8 3007.12   513.8 3006.37
   529.4    3002   581.8  3006.1   630.2 3014.81   645.9 3016.07   707.2 3029.36
#Mann= 5 ,-1,0
       0     .06       0   170.2      .1       0     227    .045       0
   265.2     .06       0   529.4      .1       0
#XS Ineff= 2 , 0
             209 3005.04     283         3005.88
Permanent Ineff=
       F       F
Bank Sta=227,265.2
XS Rating Curve= 0 ,0
Exp/Cntr(USF)=0,0
Exp/Cntr=0.5,0.3

Type RM Length L Ch R = 1 ,74079   ,218.7,251.6,284.4
BEGIN DESCRIPTION:
xs 2
END DESCRIPTION:
XS GIS Cut Line= 6
2314430.27288344611327.3666932852314398.82896813611420.650308695
2314453.33175466611507.6451410442314535.08593446611587.303059821
2314716.41251273611724.6081566612314727.94194834611916.416040033
#Sta/Elev= 30
       0 3024.14    12.6 3019.69    18.9 3016.18    31.6 3006.61    39.9 3004.52
    69.4 3005.04    81.7  3007.8    98.4    3014   120.1 3013.35   131.1 3011.93
   138.6 3009.01     152 3003.42   169.9 3002.58  212.03  2992.6   232.5 2990.97
  246.01  2992.6   260.6 2995.11   286.2 2995.94   312.2 3000.05     325 2999.69
   336.7 2997.59   356.7 2997.54   371.6 2997.64   385.9 3000.01   425.9 2998.27
   502.3 2997.63   555.3 3002.41   631.4 3009.37   695.5 3021.18   734.8 3029.82
#Mann= 9 ,-1,0
       0      .1       0    12.6     .06       0   120.1      .1       0
   138.6     .06       0  212.03    .045       0  246.01     .06       0
   385.9      .1       0   425.9     .06       0   555.3      .1       0
#XS Ineff= 2 , 0
             204    3005     253          3005.5
Permanent Ineff=
       F       F
Bank Sta=212.03,246.01
XS Rating Curve= 0 ,0
Exp/Cntr(USF)=0,0
Exp/Cntr=0.5,0.3

Type RM Length L Ch R = 1 ,73828   ,229.7,266.7,309.2
BEGIN DESCRIPTION:
xs 1
END DESCRIPTION:
XS GIS Cut Line= 4
2314430.63281414611323.9093564462314257.43393022611373.904910567
2314203.86726509611591.7426820972314236.00726417611706.018234375
#Sta/Elev= 30
       0 3024.37     4.6 3022.57    23.4 3006.74    27.5 3004.31    77.5 3003.35
    98.3 3000.36   138.7 2999.88   164.5 2998.42   197.2 2998.85   224.8 2996.69
   237.2 2997.08   253.7  2993.3   278.4 2993.45  285.41 2991.58   290.7  2990.5
  320.84 2991.61   327.8 2994.43   339.4 2996.31   352.6 2997.76     369 2997.74
   389.6 3003.88   397.8 3005.03   420.5 3003.08     431 3000.06   438.4 2999.74
   464.8 3002.15   476.7 3006.11   489.2 3008.38   516.3 3008.54   523.3 3010.05
#Mann= 5 ,-1,0
       0      .1       0      20     .06       0     120      .1       0
  285.41    .045       0  320.84      .1       0
#XS Ineff= 2 , 0
          139.53 3004.34  399.21         3006.31
Permanent Ineff=
       F       F
Bank Sta=285.41,320.84
XS Rating Curve= 0 ,0
Exp/Cntr(USF)=0,0
Exp/Cntr=0.3,0.1

Type RM Length L Ch R = 1 ,73561   ,259.8,278.3,305
XS GIS Cut Line= 2
2314476.39062589611311.6447356312313888.38940965611348.329303489
#Sta/Elev= 30
       0 3036.51    24.3 3030.22    56.3 3019.48    60.3 3016.92    72.4 3006.53
    76.4 3004.47   120.4 3003.27   132.5 3000.53   148.5 2999.32   212.9 2999.54
   252.7  2997.6   280.7 2997.32   293.5 2998.55   316.8 2998.63   348.7 2996.59
   364.9 2996.73   391.8 2995.22     426 2991.45   449.1  2990.4  457.71 2991.57
   461.9 2994.19   477.1 3010.44   481.1  3013.8   501.2 3025.31   509.2 3028.62
   529.2 3039.77   545.3 3047.62   565.3 3061.18   582.6 3069.84   589.1 3074.85
#Mann= 5 ,-1,0
       0      .1       0      60     .06       0     160      .1       0
     426    .045       0  457.71      .1       0
#XS Ineff= 2 , 0
           211.3 3006.59
Permanent Ineff=
       F       F
Bank Sta=426,457.71
XS Rating Curve= 0 ,0
Exp/Cntr(USF)=0,0
Exp/Cntr=0.3,0.1

Type RM Length L Ch R = 1 ,73283   ,182.2,184.6,186.7
XS GIS Cut Line= 3
2314481.63127844 611305.355952572314330.73930461611222.527762496
2313998.97364842610964.066542603
#Sta/Elev= 30
       0 3037.42    36.6 3025.64    70.1 3013.26    79.2 3008.91     102 3003.22
   111.2 3002.56   124.9 3003.85   147.7 3003.45   152.2 3002.88   165.9 2996.95
   190.6  2994.7   256.5 2994.89   281.9  2996.3   327.5 2995.93   337.6 2993.07
   356.6 2990.02   378.2 2989.17   395.6 2990.04   403.6 2991.98   413.7 2997.66
   444.1 3019.36   469.5 3032.03   489.8 3046.58   499.8  3050.7   515.1 3060.91
   530.3 3073.19   540.5  3078.9   565.8 3095.53   582.5 3104.84   592.7  3112.4
#Mann= 5 ,-1,0
       0      .1       0      80     .06       0  192.13      .1       0
   356.6    .045       0   395.6      .1       0
Bank Sta=356.6,395.6
XS Rating Curve= 0 ,0
Exp/Cntr(USF)=0,0
Exp/Cntr=0.3,0.1

Type RM Length L Ch R = 1 ,73098   ,68.7,294.8,336.5
BEGIN DESCRIPTION:
xs 4
END DESCRIPTION:
XS GIS Cut Line= 3
2314502.05503432611100.714918403 2314330.6417059610993.581588142
2314094.94837933610784.671594134
#Sta/Elev= 30
       0 3001.03    63.5 2995.47   112.3 2995.03   134.3  2996.9   143.7 3000.55
   157.8  3001.9   167.3  3001.7   176.7 3000.07   186.2    2995   190.9 2993.69
   216.1 2995.04   226.8 2993.63   235.3 2989.51   243.8 2988.27   283.5 2989.45
   296.3 2991.63   333.7 2990.86   340.2 2991.99   355.1 3000.03   381.8 3018.03
   391.2 3021.37     411 3033.06   419.8 3035.95   436.5 3047.14   447.9 3052.39
     456 3058.27     478 3069.63   486.2 3072.88   504.5 3083.85   517.1 3090.27
#Mann= 6 ,-1,0
       0      .1       0     100     .07       0     130     .06       0
   235.3    .045       0   283.5     .06       0  292.14      .1       0
#XS Ineff= 2 , 0
          161.58 3009.25
Permanent Ineff=
       F       F
Bank Sta=235.3,283.5
XS Rating Curve= 0 ,0
Exp/Cntr(USF)=0,0
Exp/Cntr=0.5,0.3

Type RM Length L Ch R = 1 ,72803   ,260.8,63.4,58.7
BEGIN DESCRIPTION:
xs 3
END DESCRIPTION:
XS GIS Cut Line= 6
2314616.07952744611139.8616330142314344.68644012610976.644448889
2314402.29460246610753.5810654852314441.34500336610544.128915225
2314439.56998513610501.5284778842314409.39467535610466.028113433
#Sta/Elev= 30
       0 3046.61    18.6  3038.3    59.5 3017.67    86.4 3007.64   106.8 3002.24
   173.9 2996.04   214.4 2995.16   251.9  2994.7   258.4 2995.72   270.6 3000.35
   289.3 3001.72   302.1 3000.32   316.7  2994.1   353.3 2994.94     469 2992.76
     502 2994.59   539.2 2994.76   567.9 2990.12     583 2988.42   600.5 2987.47
   633.22988.568   637.2 2990.23   645.4 2993.45   671.4 2994.01   704.4 2992.42
   805.5 2998.28   813.8 3002.95   838.9 3028.98   845.1 3032.62   849.4 3035.24
#Mann= 9 ,-1,0
       0     .06       0    18.6      .1       0   214.4     .06       0
   567.9      .1       0     583    .045       0   633.2      .1       0
   637.2     .07       0   671.4     .06       0   845.1      .1       0
#XS Ineff= 2 , 0
             573 3001.42     643         3000.55
Permanent Ineff=
       F       F
Bank Sta=583,633.2
XS Rating Curve= 0 ,0
Exp/Cntr(USF)=0,0
Exp/Cntr=0.5,0.3

Type RM Length L Ch R = 1 ,72740   ,253.1,212.6,170.5
BEGIN DESCRIPTION:
xs 2
END DESCRIPTION:
XS GIS Cut Line= 6
2314638.83504478611091.1873685882314409.25418075610988.193775814
2314424.37103324610919.1769353152314450.22009447610788.858835923
2314509.09227693610502.8289663142314428.36115651610441.138314168
#Sta/Elev= 30
       0 3038.11      58 3014.33    90.6 3003.23   108.1 2999.96     152 2996.97
     209 2994.66   307.9 2996.58   336.5 2991.47   389.6 2990.41   424.1 2991.38
   454.8 2994.63   475.2 2992.72   487.5 2993.17   503.7 2992.16   520.2 2989.61
   544.7    2991   555.7 2988.51   565.1 2987.38   584.32988.408   593.7 2989.64
   627.1 2988.93   675.3 2991.16   728.4 2989.52   753.3 2991.65   773.5 2992.18
   788.6 2995.68   798.7 2999.84   823.8 3001.31   835.5 3012.79   848.8 3022.02
#Mann= 8 ,-1,0
       0      .1       0     140     .06       0  311.62      .1       0
  412.28     .06       0  505.13     .07       0   555.7    .045       0
   584.3     .07       0  605.13     .06       0
#XS Ineff= 2 , 0
           543.7 3000.55   596.3         3000.55
Permanent Ineff=
       F       F
Bank Sta=555.7,584.3
XS Rating Curve= 0 ,0
Exp/Cntr(USF)=0,0
Exp/Cntr=0.5,0.3

Type RM Length L Ch R = 1 ,72527   ,182.4,176.9,168.9
BEGIN DESCRIPTION:
xs 1
END DESCRIPTION:
XS GIS Cut Line= 4
2314816.31280308610686.4660413952314637.75725265610527.551601509
2314484.19947927610472.1993808742314446.70281368610434.702715283
#Sta/Elev= 30
       0 2995.96    48.4 2995.15    59.1 2996.47      69 2996.78    80.2 2995.89
   116.3 2994.95   134.1 2993.36   152.4 2992.72   185.2 2993.74   200.5 2993.18
   219.7 2993.89   240.7 2993.44     245 2993.26   254.6 2991.37   270.5 2991.24
   274.7 2990.49   281.4 2987.95   293.2 2987.51   310.9 2987.99   317.2 2989.85
   320.3 2990.01   334.3 2990.13   348.4  2989.2   376.5 2991.14   393.8 2991.34
     408 2994.35   419.3 2999.45   423.5 3000.24   453.2 3000.21   455.3 3000.69
#Mann= 4 ,-1,0
       0      .1       0   281.4    .045       0   310.9      .1       0
  369.03     .06       0
Bank Sta=281.4,310.9
XS Rating Curve= 0 ,0
Exp/Cntr(USF)=0,0
Exp/Cntr=0.3,0.1

Type RM Length L Ch R = 1 ,72350   ,341.2,333.1,323
XS GIS Cut Line= 4
2315040.08109113 610295.575837582314780.13825665610352.528000169
 2314480.7656503610327.8541654632314370.34427445610448.277931208
#Sta/Elev= 30
       0 3012.18    16.3 3012.07    65.4 3003.97   114.6  2999.2   172.6 2996.53
   241.5 2996.08     262 2993.93   338.3 2992.67   358.4 2990.71   378.5 2991.43
   402.5 2989.25   458.7 2989.18   463.42987.529   470.8  2986.2   495.4 2986.27
   501.2 2987.54   510.9 2990.61   533.6 2990.56     555 2992.99   578.5 2993.67
   595.4 2998.25   624.5 2999.42   638.4 2998.85   644.3 3001.88   652.8 3008.78
   664.1 3022.59   676.8 3033.03   706.6 3044.58   717.9 3046.91   729.9 3052.06
#Mann= 6 ,-1,0
       0     .06       0      40      .1       0   463.4    .045       0
   501.2      .1       0   596.5     .06       0   666.5      .1       0
#XS Ineff= 2 , 0
                          554.03         2996.94
Permanent Ineff=
       F       F
Bank Sta=463.4,501.2
XS Rating Curve= 0 ,0
Exp/Cntr(USF)=0,0
Exp/Cntr=0.3,0.1

Type RM Length L Ch R = 1 ,72017   ,407.5,358.5,314
XS GIS Cut Line= 6
2314863.24785012609931.814317962  2314784.172804610007.954949745
2314768.27565204 610013.099413062314511.73423848610056.582260237
2314373.21975032610169.127988112 2314355.7877797610426.308557644
#Sta/Elev= 30
       0 3017.82    15.4 3012.31      32 3009.51      71 2999.72    98.7 2994.86
   201.52986.089   219.3 2985.19   242.2 2986.05   248.3  2988.5   280.8  2988.2
   288.9 2990.88     297 2991.44   378.1  2989.7   427.3 2991.61   476.4 2990.57
   509.8 2991.97   597.3 2992.21   625.3 2997.93   637.4 2997.52   667.6 2991.66
   690.1 2991.68   709.5 2996.58   725.6 2998.03   733.6 3001.11   753.3 3012.38
   769.7  3023.9   785.7 3030.64   793.7 3032.34   805.8    3039   822.9 3044.88
#Mann= 6 ,-1,0
       0     .06       0      40      .1       0   201.5    .045       0
   242.2      .1       0  536.68     .06       0  745.16      .1       0
#XS Ineff= 2 , 0
                          511.32            2996
Permanent Ineff=
       F       F
Bank Sta=201.5,242.2
XS Rating Curve= 0 ,0
Exp/Cntr(USF)=0,0
Exp/Cntr=0.3,0.1

Type RM Length L Ch R = 1 ,71659   ,191.3,190.2,189.5
XS GIS Cut Line= 3
2314402.06392607609718.6949580422314375.28059351610049.022726345
 2314342.7916704 610429.17616217
#Sta/Elev= 30
       0  3080.9    34.6 3061.16    52.3 3047.02    74.6  3044.8    78.3 3042.83
    98.8 3027.03   122.9 3013.12     151 2991.09   163.7 2985.29   171.1 2983.97
   205.9 2985.17   214.6 2986.64   227.2 2986.12   243.3 2988.48   255.3 2987.31
   279.4 2988.89   303.5 2988.37   323.5 2991.42   367.9 2990.22   399.8 2991.92
   476.1  2992.2   500.9 2997.77     512 2997.57   547.7 2991.38   576.5 2991.44
   596.5 2996.65   608.6 2997.41   616.6 2999.79   648.8 3020.13     713 3047.12
#Mann= 7 ,-1,0
       0      .1       0      40     .06       0     140      .1       0
   163.7    .045       0   205.9      .1       0  441.41     .06       0
  631.41      .1       0
#XS Ineff= 2 , 0
                          324.88         2993.86
Permanent Ineff=
       F       F
Bank Sta=163.7,205.9
XS Rating Curve= 0 ,0
Exp/Cntr(USF)=0,0
Exp/Cntr=0.3,0.1

Type RM Length L Ch R = 1 ,71468   ,218.3,217.2,219.2
XS GIS Cut Line= 2
2314207.04259798609704.5452959632314169.76721531 610421.65265787
#Sta/Elev= 30
       0 3084.34    36.7 3062.89    60.7 3044.71    84.7 3041.66   104.8 3022.64
   112.8 3017.16   156.8 2989.22   170.9 2983.59   192.9 2982.79   201.3 2983.53
     237 2985.13   263.8 2984.53   280.7 2986.15     301 2984.86   317.1 2987.56
   333.1 2986.66   345.1  2988.5   357.1 2987.57   373.1 2994.66   381.1 2995.77
   389.2 2994.93   409.2 2988.99   496.2 2990.97   525.3 2989.56   553.4 2990.95
   573.4 2989.64   597.4 2990.49   609.5 2994.23   639.8 3010.85   718.1 3045.23
#Mann= 7 ,-1,0
       0      .1       0      60     .06       0     160      .1       0
   170.9    .045       0   201.3      .1       0     250     .06       0
     450      .1       0
#XS Ineff= 2 , 0
                           384.9         3002.61
Permanent Ineff=
       F       F
Bank Sta=170.9,201.3
XS Rating Curve= 0 ,0
Exp/Cntr(USF)=0,0
Exp/Cntr=0.3,0.1

Type RM Length L Ch R = 1 ,71251   ,318.6,319.8,320.7
XS GIS Cut Line= 2
2314009.24171512609706.1960695112314003.88504861610393.634938683
#Sta/Elev= 30
       0 3088.49      19 3075.33      47 3060.08    78.5 3037.04      99  3035.2
     103 3033.61     115 3023.21     127 3015.25   158.8 2996.47     179  2985.9
     187 2984.17     239 2985.27   255.9 2982.94     271 2981.77     287 2981.81
  291.67 2982.98     299  2988.1     315 2988.75     331 2994.24     343 2993.66
     359  2987.3     375 2986.83     403 2988.79     415 2987.99     487 2988.28
     607 2990.53   630.9 2997.87     655 3008.74   674.8 3015.84   687.5 3022.68
#Mann= 7 ,-1,0
       0      .1       0      60     .06       0     150      .1       0
   255.9    .045       0  291.67      .1       0     350     .06       0
     450      .1       0
#XS Ineff= 2 , 0
                          333.63         3003.52
Permanent Ineff=
       F       F
Bank Sta=255.9,291.67
XS Rating Curve= 0 ,0
Exp/Cntr(USF)=0,0
Exp/Cntr=0.3,0.1

Type RM Length L Ch R = 1 ,70932   ,225.3,248.8,270.1
XS GIS Cut Line= 3
2313755.30816176609692.0504053762313706.48745922609827.021553318
2313657.53049425610413.874783569
#Sta/Elev= 30
       0 3070.96      31 3059.92    52.2 3040.44      65  3031.4      82 3031.58
    90.8 3029.84     116 3006.28   145.7 2988.24   153.7 2985.59   161.7 2986.14
   173.6 2983.75   199.5 2982.47   214.4 2980.88   250.1 2980.95   260.8  2982.4
   278.2 2982.59   290.2 2985.26   310.3 2986.38   330.3 2982.97   342.4 2982.65
   346.4    2983   362.4 2989.85   370.5  2990.9   394.6 2984.93   615.3 2989.11
   651.5 2998.14   675.5 3010.05   699.6 3018.58   711.7 3020.81   732.4 3028.85
#Mann= 7 ,-1,0
       0      .1       0      70     .06       0  173.53      .1       0
   199.5    .045       0   260.8      .1       0  373.53     .06       0
  473.53      .1       0
#XS Ineff= 2 , 0
                          371.83         2996.58
Permanent Ineff=
       F       F
Bank Sta=199.5,260.8
XS Rating Curve= 0 ,0
Exp/Cntr=0.3,0.1

Type RM Length L Ch R = 1 ,70683   ,409.5,432.8,448.8
XS GIS Cut Line= 4
2313699.37552126609635.0267261852313544.11392241609715.636294428
2313341.52066214610013.3643968572313240.10160925610247.135194623
#Sta/Elev= 30
       0 3052.67     8.1 3051.08    21.6 3044.26    39.7 3031.58    66.3 3028.85
    80.2 3020.69   134.9  3004.6   156.8 2993.13   174.9  2986.1     201  2983.8
   244.5  2985.9   262.4  2980.8   268.7 2980.06   292.12980.861   307.4 2983.62
   331.6 2984.12   438.1 2983.69   447.7 2981.37     510 2980.83   525.2 2986.85
   534.8 2988.38   543.6  2987.7   557.2 2981.46   604.6 2981.27     615 2983.17
   648.5 2982.09     670 2986.76   722.3  2992.3   757.2 3003.12   789.9 3016.82
#Mann= 7 ,-1,0
       0     .06       0      80      .1       0   262.4    .045       0
   292.1      .1       0  374.94     .08       0  464.94     .06       0
  585.06      .1       0
#XS Ineff= 2 , 0
                          536.34         2997.19
Permanent Ineff=
       F       F
Bank Sta=262.4,292.1
XS Rating Curve= 0 ,0
Exp/Cntr(USF)=0,0
Exp/Cntr=0.3,0.1

Type RM Length L Ch R = 1 ,70250   ,276,276.9,269.2
XS GIS Cut Line= 3
2313696.33997094609622.3363808632313266.80140561609722.578477749
2312874.00611457609815.981936251
#Sta/Elev= 30
       0 3052.27    20.7 3042.58    37.1 3031.18    57.7 3029.55      70 3021.78
    98.2  3011.3   135.7 2993.81   160.4 2985.46   193.2  2985.5     219 2982.93
   242.3 2984.85   316.4 2983.31   443.8 2984.95   493.1 2979.45     526  2981.5
     565 2979.47   583.6 2978.12   590.6 2979.58     600 2984.68   612.4 2987.51
   620.6  2986.8   632.9 2982.04   678.5 2981.62   686.4 2985.25   706.9 3000.39
   723.4 3010.16   764.8 3024.82   780.9 3033.56   805.6 3043.41   844.8 3068.28
#Mann= 7 ,-1,0
       0     .06       0      70      .1       0     380     .08       0
  481.08      .1       0     565    .045       0   590.6     .06       0
  681.08      .1       0
#XS Ineff= 2 , 0
                          612.96         2996.03
Permanent Ineff=
       F       F
Bank Sta=565,590.6
XS Rating Curve= 0 ,0
Exp/Cntr(USF)=0,0
Exp/Cntr=0.3,0.1

Type RM Length L Ch R = 1 ,69973   ,326.6,328.7,328.9
XS GIS Cut Line= 5
 2313660.6856953609539.6135527992313436.91071832609591.256458123
2313318.11784545609547.7548427072313023.10544355 609576.74398394
2312874.00391285609555.443765269
#Sta/Elev= 30
       0 3036.56    16.9 3027.28    33.4 3026.31      58 3009.35    81.8 2996.68
   111.4 2985.07   193.5 2983.44   234.7 2985.09   253.7 2982.34   290.1 2983.49
   315.6 2980.81   358.1 2984.13   406.3 2981.97   414.2 2979.32   419.1 2977.74
   457.92979.274   498.8 2981.24   583.2 2981.06   603.3 2987.44   627.4 2989.78
   643.5  2997.5   659.6 3007.95   671.7 3019.25   732.3 3056.54   746.1 3068.38
   756.6 3072.47   772.7 3083.23   780.8  3089.6   792.9 3104.89   803.2 3110.22
#Mann= 9 ,-1,0
       0     .06       0      40      .1       0  239.66     .08       0
  329.66      .1       0  339.66     .08       0   414.2    .045       0
   457.9      .1       0  546.16     .06       0  636.16      .1       0
#XS Ineff= 2 , 0
          236.62 2996.38
Permanent Ineff=
       F       F
Bank Sta=414.2,457.9
XS Rating Curve= 0 ,0
Exp/Cntr(USF)=0,0
Exp/Cntr=0.3,0.1

Type RM Length L Ch R = 1 ,69644   ,286.8,287.6,287.4
XS GIS Cut Line= 3
 2313617.2498918609214.1606513992313149.35931303609240.645822693
2312983.96052786609173.352654899
#Sta/Elev= 30
       0 3025.67    17.1 3017.64    29.1 3017.57    37.1 3016.03    57.2 3002.83
    85.2 2992.31   137.3 2984.53   189.4  2983.8   201.4 2980.47   237.5 2980.11
   249.5 2982.34   277.5 2978.72   345.6 2980.68   369.7 2978.46   389.7 2978.41
   393.7 2977.16   401.7  2976.4   426.9 2977.15   445.8 2984.55   474.2 2987.37
   482.9 2996.74   513.1 3033.03   526.1 3038.09   543.3 3052.85   556.3 3056.71
   569.2  3067.2   586.5 3078.33   607.3  3089.4     634 3109.42   647.2 3116.84
#Mann= 6 ,-1,0
       0     .06       0      90      .1       0     390     .06       0
   393.7    .045       0   426.9     .06       0  588.64      .1       0
Bank Sta=393.7,426.9
XS Rating Curve= 0 ,0
Exp/Cntr(USF)=0,0
Exp/Cntr=0.3,0.1

Type RM Length L Ch R = 1 ,69357   ,313.8,301,285.5
XS GIS Cut Line= 2
2313660.33698544608985.6629158342313055.05577155608964.362697163
#Sta/Elev= 30
       0  3054.4    32.2 3040.71    80.2  3024.8    95.1 3017.22   104.2 3010.64
   124.2 3008.41   140.2 2998.38   156.3  2991.5   192.3 2984.51   224.3 2983.47
   240.3 2978.59   288.3 2979.49   316.4 2978.37   323.2 2976.48   328.4 2975.16
   356.3 2975.03   368.9 2976.47   384.4 2979.61   408.4 2980.29   420.4 2985.17
   448.4 2985.43   452.4 2987.29     456 2990.77   464.4 3002.18   476.7 3013.39
   504.5 3029.71   520.5 3040.99   532.5 3045.43   576.7 3069.33   605.7 3075.95
#Mann= 7 ,-1,0
       0      .1       0      30     .06       0     130      .1       0
   323.2    .045       0   368.9      .1       0     430     .06       0
     530      .1       0
Bank Sta=323.2,368.9
XS Rating Curve= 0 ,0
Exp/Cntr(USF)=0,0
Exp/Cntr=0.3,0.1
